HEC-RAS study US278overBeaver.prj: US 278 over Beaver Dam Cr_Prelim

--- US278overBeaver.g06 (geometry) --- (continued)

Type RM Length L Ch R = 4 ,14763.71,,,
Bridge Culvert--1,0,-1,-1, 0
Deck Dist Width WeirC Skew NumUp NumDn MinLoCord MaxHiCord MaxSubmerge Is_Ogee
32,30,2.6,0, 60, 60, , , 0.98, 0, 0,0,,
       0   63.78    81.7   99.81  162.22  186.05  197.95  210.94  255.53  260.33
  272.37  300.48  369.93  390.87  404.19  414.57  429.67   535.5  547.58  562.45
  566.78  592.29  614.78  627.37  655.63  708.77  718.15  731.21  735.25  736.79
  764.32  775.26  795.89  803.45  820.64  841.84  876.75  977.36 1029.02 1079.76
 1096.75 1119.48 1151.72  1159.2 1165.72 1172.95 1196.52 1233.91 1320.17 1398.01
 1412.77 1423.47 1451.06 1465.93 1467.23 1468.18 1468.69 1469.53 1473.91 1506.19
   60.12   58.83   58.68   58.13    57.2   56.38   56.41   56.03   55.28   55.02
   54.87   54.15   52.87   52.15   52.15   51.79   51.76   50.37   50.39   49.91
   50.01   49.72   49.76   49.33   49.52   49.37   49.13   49.28   49.15   49.27
   49.03   49.23   49.24   49.04   48.94   49.14   49.09   49.58   50.69   51.35
   51.73   52.55   53.34   53.75   53.73   54.12   54.84   56.62   59.94   63.34
   64.14   64.45   65.87   66.41    66.3   66.35   66.59   66.49   66.79   68.13
                                                                                
                                                                                
                                                                                
                                                                                
                                                                                
                                                                                
       0   63.78    81.7   99.81  162.22  186.05  197.95  210.94  255.53  260.33
  272.37  300.48  369.93  390.87  404.19  414.57  429.67   535.5  547.58  562.45
  566.78  592.29  614.78  627.37  655.63  708.77  718.15  731.21  735.25  736.79
  764.32  775.26  795.89  803.45  820.64  841.84  876.75  977.36 1029.02 1079.76
 1096.75 1119.48 1151.72  1159.2 1165.72 1172.95 1196.52 1233.91 1320.17 1398.01
 1412.77 1423.47 1451.06 1465.93 1467.23 1468.18 1468.69 1469.53 1473.91 1506.19
   60.12   58.83   58.68   58.13    57.2   56.38   56.41   56.03   55.28   55.02
   54.87   54.15   52.87   52.15   52.15   51.79   51.76   50.37   50.39   49.91
   50.01   49.72   49.76   49.33   49.52   49.37   49.13   49.28   49.15   49.27
   49.03   49.23   49.24   49.04   48.94   49.14   49.09   49.58   50.69   51.35
   51.73   52.55   53.34   53.75   53.73   54.12   54.84   56.62   59.94   63.34
   64.14   64.45   65.87   66.41    66.3   66.35   66.59   66.49   66.79   68.13
                                                                                
                                                                                
                                                                                
                                                                                
                                                                                
                                                                                
BR Coef=-1 , 0 , 0 ,, 0 ,,,0.8,-1,,0,
WSPro=,,,, 1 ,,,, 0 ,,,, 0 ,,,,-1 ,-1 ,-1 , 0 , 0 , 0 , 0 , 0
Multiple Barrel Culv=2,12,10,36,0.013,0.4,1,8,1,38.8,38.75, 2,Culvert #1  , 0 ,32
   989.5  989.54 1000.56  1000.5
BC Culvert Barrel=1,Barrel #1,0
BC Culvert Barrel=2,Barrel #2,0
Culvert Bottom n=0.013
Multiple Barrel Culv=2,12,10,36,0.013,0.4,1,8,1,39,38.95, 2,Culvert #2  , 0 ,32
  1035.5  1035.5  1046.5  1046.5
BC Culvert Barrel=1,Barrel #1,0
BC Culvert Barrel=2,Barrel #2,0
Culvert Bottom n=0.013
BC Mult= 2 ,0,1030.15,0,1030.15
BC Mult= 2 ,1009.11,1508.37,1009.11,1508.37
BC Design=,, 0 ,, 0 ,,,,,,
BC Use User HTab Curves=0
BC User HTab FreeFlow(D)= 0

--- US278overBeaver.g07 (geometry) ---

Geom Title=Prop Cond_Culv_Double 10x8+Double10x12
Program Version=6.50

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
River Reach=Beaver Dam Creek,Reach 1

Type RM Length L Ch R = 4 ,14763.71,,,
Bridge Culvert--1,0,-1,-1, 0
Deck Dist Width WeirC Skew NumUp NumDn MinLoCord MaxHiCord MaxSubmerge Is_Ogee
32,30,2.6,0, 60, 60, , , 0.98, 0, 0,0,,
       0   63.78    81.7   99.81  162.22  186.05  197.95  210.94  255.53  260.33
  272.37  300.48  369.93  390.87  404.19  414.57  429.67   535.5  547.58  562.45
  566.78  592.29  614.78  627.37  655.63  708.77  718.15  731.21  735.25  736.79
  764.32  775.26  795.89  803.45  820.64  841.84  876.75  977.36 1029.02 1079.76
 1096.75 1119.48 1151.72  1159.2 1165.72 1172.95 1196.52 1233.91 1320.17 1398.01
 1412.77 1423.47 1451.06 1465.93 1467.23 1468.18 1468.69 1469.53 1473.91 1506.19
   60.12   58.83   58.68   58.13    57.2   56.38   56.41   56.03   55.28   55.02
   54.87   54.15   52.87   52.15   52.15   51.79   51.76   50.37   50.39   49.91
   50.01   49.72   49.76   49.33   49.52   49.37   49.13   49.28   49.15   49.27
   49.03   49.23   49.24   49.04   48.94   49.14   49.09   49.58   50.69   51.35
   51.73   52.55   53.34   53.75   53.73   54.12   54.84   56.62   59.94   63.34
   64.14   64.45   65.87   66.41    66.3   66.35   66.59   66.49   66.79   68.13
                                                                                
                                                                                
                                                                                
                                                                                
                                                                                
                                                                                
       0   63.78    81.7   99.81  162.22  186.05  197.95  210.94  255.53  260.33
  272.37  300.48  369.93  390.87  404.19  414.57  429.67   535.5  547.58  562.45
  566.78  592.29  614.78  627.37  655.63  708.77  718.15  731.21  735.25  736.79
  764.32  775.26  795.89  803.45  820.64  841.84  876.75  977.36 1029.02 1079.76
 1096.75 1119.48 1151.72  1159.2 1165.72 1172.95 1196.52 1233.91 1320.17 1398.01
 1412.77 1423.47 1451.06 1465.93 1467.23 1468.18 1468.69 1469.53 1473.91 1506.19
   60.12   58.83   58.68   58.13    57.2   56.38   56.41   56.03   55.28   55.02
   54.87   54.15   52.87   52.15   52.15   51.79   51.76   50.37   50.39   49.91
   50.01   49.72   49.76   49.33   49.52   49.37   49.13   49.28   49.15   49.27
   49.03   49.23   49.24   49.04   48.94   49.14   49.09   49.58   50.69   51.35
   51.73   52.55   53.34   53.75   53.73   54.12   54.84   56.62   59.94   63.34
   64.14   64.45   65.87   66.41    66.3   66.35   66.59   66.49   66.79   68.13
                                                                                
                                                                                
                                                                                
                                                                                
                                                                                
                                                                                
BR Coef=-1 , 0 , 0 ,, 0 ,,,0.8,-1,,0,
WSPro=,,,, 1 ,,,, 0 ,,,, 0 ,,,,-1 ,-1 ,-1 , 0 , 0 , 0 , 0 , 0
Multiple Barrel Culv=2,8,10,36,0.013,0.4,1,8,1,38.8,38.75, 2,Culvert #1  , 0 ,32
   989.5  989.54 1000.56  1000.5
BC Culvert Barrel=1,Barrel #1,0
BC Culvert Barrel=2,Barrel #2,0
Culvert Bottom n=0.013
Multiple Barrel Culv=2,12,10,36,0.013,0.4,1,8,1,39,38.95, 2,Culvert #2  , 0 ,32
  1035.5  1035.5  1046.5  1046.5
BC Culvert Barrel=1,Barrel #1,0
BC Culvert Barrel=2,Barrel #2,0
Culvert Bottom n=0.013
BC Mult= 2 ,0,1030.15,0,1030.15
BC Mult= 2 ,1009.11,1508.37,1009.11,1508.37
BC Design=,, 0 ,, 0 ,,,,,,
BC Use User HTab Curves=0
BC User HTab FreeFlow(D)= 0
